HEC-RAS study wekiva_ras.prj: wekiva_ras

--- wekiva_ras.g01 (geometry) --- (continued)

Type RM Length L Ch R = 1 ,318.81  ,61.1549,61.1549,61.1549
BEGIN DESCRIPTION:
MFL_SR46B
END DESCRIPTION:
Node Name=MFL_SR46B
XS GIS Cut Line= 2
 458972.529304883187577.41857002459149.2051048793187568.68737002
#Sta/Elev= 30
       0   17.26   12.98   12.39      30    7.85     105    8.19     155    7.81
     175    8.26     208     6.9     215    5.96     235     .96     255     .36
     262    -.34     285    -.54     295   -1.64     313     .46     325    4.96
     335    2.56     375    2.16     385     .46     395    -.04     405     .26
     430    7.02     435    7.52     467    7.78     495    6.96     535    7.43
  552.12    11.2  564.22   18.16  574.11   22.41  588.18   23.35  633.37   23.11
#Mann= 3 , 0 , 0
       0     .22       0     175      .2       0     435     .22       0
Bank Sta=175,435
XS Rating Curve= 0 ,0
Exp/Cntr=0.5,0.3

Type RM Length L Ch R = 3 ,318.50  ,,,
BEGIN DESCRIPTION:
SR46
SR46
END DESCRIPTION:
Bridge Culvert--1,0,-1,-1, 0
Deck Dist Width WeirC Skew NumUp NumDn MinLoCord MaxHiCord MaxSubmerge Is_Ogee
10,42,2.6,0, 2, 2, , , 0.98, 0, 0,0,,
       0    1000
   22.41   22.41
   16.66   16.66
       0    1000
   22.41   22.41
   16.66   16.66
Pier Skew, UpSta & Num, DnSta & Num=  ,47.6, 2 ,70.62, 2 , 0 , 0 , 0 ,,
    2.51    2.51
      -5      20
    2.51    2.51
      -5      20
Pier Skew, UpSta & Num, DnSta & Num=  ,98.58, 2 ,121.24, 2 , 0 , 0 , 0 ,,
    2.59    2.59
      -5      20
    2.59    2.59
      -5      20
Pier Skew, UpSta & Num, DnSta & Num=  ,149.66, 2 ,172.34, 2 , 0 , 0 , 0 ,,
    2.76    2.76
      -5      20
    2.76    2.76
      -5      20
Pier Skew, UpSta & Num, DnSta & Num=  ,200.99, 2 ,223.47, 2 , 0 , 0 , 0 ,,
    2.49    2.49
      -5      20
    2.49    2.49
      -5      20
Pier Skew, UpSta & Num, DnSta & Num=  ,251.54, 2 ,274.63, 2 , 0 , 0 , 0 ,,
    2.88    2.88
      -5      20
    2.88    2.88
      -5      20
Pier Skew, UpSta & Num, DnSta & Num=  ,302.68, 2 ,325.54, 2 , 0 , 0 , 0 ,,
    2.56    2.56
      -5      20
    2.56    2.56
      -5      20
Pier Skew, UpSta & Num, DnSta & Num=  ,353.48, 2 ,376.5, 2 , 0 , 0 , 0 ,,
    2.72    2.72
      -5      20
    2.72    2.72
      -5      20
Pier Skew, UpSta & Num, DnSta & Num=  ,404.98, 2 ,427.78, 2 , 0 , 0 , 0 ,,
    2.97    2.97
      -5      20
    2.97    2.97
      -5      20
Pier Skew, UpSta & Num, DnSta & Num=  ,455.88, 2 ,478.66, 2 , 0 , 0 , 0 ,,
     2.7     2.7
      -5      20
     2.7     2.7
      -5      20
Pier Skew, UpSta & Num, DnSta & Num=  ,506.88, 2 ,529.66, 2 , 0 , 0 , 0 ,,
    2.41    2.41
      -5      20
    2.41    2.41
      -5      20
BR Coef=-1 , 0 , 0 ,, 0 ,,,0.8,-1,,0,
WSPro=,,,, 1 ,,,, 0 ,,,, 0 ,,,,-1 ,-1 ,-1 , 0 , 0 , 0 , 0 , 0
BR U #Sta/Elev= 44
       0   17.26   12.98   12.39   27.84    8.14   48.09    7.78   69.88     7.9
   91.84    7.83  112.66     7.9  135.55     7.9  156.96    7.81  178.43    7.65
     199    7.69  203.01    7.17   207.4    6.39  211.42    5.77  218.91     2.7
  229.06    2.75  243.78    1.06  262.24     .89  278.06       0   291.9    -.65
  304.49    -.04  318.13    1.89  327.16    1.97  344.52    2.07  357.51    2.42
  374.28     1.7  385.06     .05  400.25    -.24  412.27    1.12  425.87    5.45
  427.42    6.37   432.1    7.01  437.69    7.74  457.24    7.43  476.77    7.13
   498.1    7.04  517.84    7.12  536.57    7.77  552.12    11.2  564.22   18.16
  574.11   22.41  588.18   23.35  609.46   23.25  633.37   23.11
BR U #Mann= 4
       0     .95   27.84    .035     199      .2  437.69    .035
BR U Banks=199,437.69
BR D #Sta/Elev= 49
       0   10.35      21    9.08   41.65     8.4   64.58    7.75   85.98    7.97
  106.38    8.07  125.87    8.33   145.7    8.71  168.11    9.27  192.29   10.09
  210.25    8.74  220.12    7.59  227.57     7.1  236.37    6.38  238.32     6.1
   245.7    4.92   254.2    2.68  263.47     .67  275.36     .81  288.97     .94
  304.74    1.89  322.23    3.58  341.07    4.31  362.87     3.7  363.01    3.72
  382.62    3.52  394.53    2.25  403.96      .8  419.02     .97  428.68    3.53
   440.6    6.16  441.37    6.38  448.17    6.98  459.02     7.5  475.81    8.31
  492.99    8.37  512.85    8.63  533.41    8.87  552.15    8.66  564.21    8.81
   573.9   10.85  583.12   13.93  589.65   18.13  596.63    22.1  607.62   23.11
  623.77   22.89  642.57   22.72   660.5   22.75  679.02    22.8
BR D #Mann= 3
       0      .5  210.25      .2  475.81     .95
BR D Banks=192.29,475.81
BC Design=,, 0 ,, 0 ,,,,,,
BC HTab HWMax=16.66
BC Use User HTab Curves=0
BC User HTab FreeFlow(D)= 0

Type RM Length L Ch R = 1 ,318.19  ,16.1745,16.1745,16.1745
BEGIN DESCRIPTION:
MFL_SR46A
END DESCRIPTION:
Node Name=MFL_SR46A
XS GIS Cut Line= 3
 458972.715004883187593.78647002459149.7894048793187585.95147002
459323.6393266723187578.25914331
#Sta/Elev= 30
       0   10.35      52    7.63      87    8.22     157    8.48     167    9.15
     184     9.3     207     8.9     227    7.42     247    4.76     257    2.16
     267     .76     286     .36     307    1.46     327    3.36     357    4.56
     377    3.76     387    1.96     397    1.16     417    1.16     427    2.71
     439    5.66     448    7.05  486.94    8.24     557    8.28  564.21    8.81
   573.9   10.85  583.12   13.93  596.63    22.1  607.62   23.11  679.02    22.8
#Mann= 3 , 0 , 0
       0     .22       0     184      .2       0  486.94     .22       0
Bank Sta=184,486.94
XS Rating Curve= 0 ,0
Exp/Cntr=0.5,0.3

Type RM Length L Ch R = 1 ,318.03  ,78.5761,78.5761,78.5761
BEGIN DESCRIPTION:
XS9
END DESCRIPTION:
Node Name=XS9
XS GIS Cut Line= 2
 458968.757504883187600.67747002459170.9561048793187586.74517002
#Sta/Elev= 30
       0   10.35      21    9.08   64.58    7.75  125.87    8.33  192.29   10.09
  236.37    6.38   245.7    4.92   254.2    2.68  263.47     .67  288.97     .94
  304.74    1.89  322.23    3.58  341.07    4.31  382.62    3.52  394.53    2.25
  403.96      .8  419.02     .97  428.68    3.53  441.37    6.38  448.17    6.98
  475.81    8.31  533.41    8.87  564.21    8.81   573.9   10.85  583.12   13.93
  589.65   18.13  596.63    22.1  607.62   23.11  642.57   22.72  679.02    22.8
#Mann= 3 , 0 , 0
       0     .22       0  192.29      .2       0  475.81     .22       0
Bank Sta=192.29,475.81
XS Rating Curve= 0 ,0
Exp/Cntr=0.5,0.3

Type RM Length L Ch R = 1 ,317.25  ,143.1102,143.1102,143.1102
BEGIN DESCRIPTION:
MFL_SR46F
END DESCRIPTION:
Node Name=MFL_SR46F
#Sta/Elev= 30
 -150.52    14.3   20.95     7.8  190.85    5.86  226.96    6.78     406    6.63
     417    5.04     422    3.54     427     .04     442   -3.66     447   -3.66
     452   -1.76     462    -.56     472    -.76     487     .74     507    4.64
     517    5.64     522    7.45     577    7.25     582    5.34     592    2.94
     607     .44     632    1.74     672    6.64   716.2     7.1  717.87    7.98
   763.1    6.66  817.89    7.07  878.48    9.23   897.8   10.27  905.78   11.67
#Mann= 3 , 0 , 0
 -150.52     .22       0     406      .2       0     522     .22       0
#XS Ineff= 1 ,-1
  157.53  206.53    6.67
Permanent Ineff=
       F
Bank Sta=406,522
XS Rating Curve= 0 ,0
Exp/Cntr=0.3,0.1

Type RM Length L Ch R = 1 ,315.81  ,997.3753,997.3753,997.3753
BEGIN DESCRIPTION:
XS8
XS8
END DESCRIPTION:
Node Name=XS8
XS GIS Cut Line= 2
 458917.374004883187636.49117002 459187.742604883187689.83957002
#Sta/Elev= 30
 -150.52    14.3       0    8.29   63.91    7.24  157.53    6.69  190.85    5.86
  206.53    6.67  325.03    6.67  365.22    7.06     366    7.63  421.89    -.44
  450.99     .06  477.02    2.51  490.39     5.5  494.86    7.36  527.01    6.67
  585.88    6.73  594.18    8.08  608.44    6.77   621.6    2.26  633.11    1.05
  673.47     2.5   684.5    2.05  698.82    3.28   716.2     7.1  717.87    7.98
  748.38    6.81   798.6    6.66  878.48    9.23   897.8   10.27  905.78   11.67
#Mann= 3 , 0 , 0
 -150.52     .22       0     366      .2       0  494.86     .22       0
#XS Ineff= 1 ,-1
  157.53  206.53    6.67
Permanent Ineff=
       F
Bank Sta=366,494.86
XS Rating Curve= 0 ,0
Exp/Cntr=0.3,0.1

Type RM Length L Ch R = 1 ,305.84  ,30.4134,30.4134,30.4134
BEGIN DESCRIPTION:
XS7
END DESCRIPTION:
Node Name=XS7
XS GIS Cut Line= 2
458912.9379048793188032.57667002 459199.229404883187905.09737002
#Sta/Elev= 30
       0   10.14  177.56    7.82  318.03    6.89  372.37    7.87  375.96    7.37
  378.14    4.98  399.46    3.24  420.29    4.03     457    3.46  507.07    4.16
   542.5     3.3  579.19    4.34  689.43     3.9  710.74    4.72  717.21    6.29
  733.55    7.32  741.28     6.3  743.89    3.82  775.54     .63  797.98    7.13
  805.16    7.82  810.18    6.94  876.64    6.23  891.82    2.76  902.61    1.94
  928.63    3.05  942.04    5.31  945.29    7.68  948.81    8.82 1032.06   11.73
#Mann= 5 , 0 , 0
       0     .22       0  177.56     .22       0  372.37      .2       0
  733.55     .22       0  805.16     .22       0
#XS Ineff= 1 ,-1
  805.16  945.29    7.82
Permanent Ineff=
       F
Bank Sta=372.37,733.55
XS Rating Curve= 0 ,0
Exp/Cntr=0.3,0.1

Type RM Length L Ch R = 1 ,305.54  ,1330.971,1330.971,1330.971
BEGIN DESCRIPTION:
MFL_Maple
END DESCRIPTION:
Node Name=MFL_Maple
XS GIS Cut Line= 4
458874.819588939 3188076.6633844 459012.990904883188004.24317002
459034.858588939 3187992.7815844459109.3117230033187953.75820322
#Sta/Elev= 30
    -156   18.03     -32   11.02     188    7.89  372.37    6.96     377    6.85
     383    4.77     403    3.17     523    4.27     708    4.17     718    5.07
     723    6.82  733.55    7.05   745.5    6.87     748    4.17     753    3.07
     773    1.17     783    1.37     800    7.52     803    7.79     820    7.79
     828    6.49     875    5.92     888    2.92     893     .27     898       0
     903    1.18     933     2.7     938    3.97     948     8.6 1032.06   11.73
#Mann= 6 , 0 , 0
    -156     .22       0     188     .22       0  372.37      .2       0
  733.55     .22       0     773     .22       0     803     .22       0
#XS Ineff= 1 ,-1
  805.16  945.29    7.82
Permanent Ineff=
       F
Bank Sta=372.37,733.55
XS Rating Curve= 0 ,0
Exp/Cntr=0.3,0.1

Type RM Length L Ch R = 1 ,292.23  ,1556.693,1556.693,1556.693
BEGIN DESCRIPTION:
XS6
END DESCRIPTION:
Node Name=XS6
XS GIS Cut Line= 2
 459066.962404883188398.80067002 459329.354904883188309.45017002
#Sta/Elev= 30
  -82.59   12.48   20.95    7.37   90.95    6.47  131.64    5.37  170.22    6.86
  175.34    5.34  221.51    6.67  262.91     6.7  312.35    3.93  347.42     4.7
  364.26    4.22  382.29    4.82  385.58    7.16  414.57    8.55  419.68       6
  420.26    4.72  425.41     3.1  488.98    3.77  683.22    2.93  703.84    3.89
  725.17    3.03  742.68    3.96  756.14     6.2  756.48    5.44  763.62    8.22
  768.16    7.42  783.48    8.14  828.24    8.18   921.8    9.53 1008.19    12.8
#Mann= 4 , 0 , 0
  -82.59     .22       0   90.95     .22       0  414.57      .2       0
  763.62     .22       0
Bank Sta=414.57,763.62
XS Rating Curve= 0 ,0
Exp/Cntr=0.3,0.1

Type RM Length L Ch R = 1 ,276.66  ,2392.52,2392.52,2392.52
BEGIN DESCRIPTION:
XS5
END DESCRIPTION:
Node Name=XS5
XS GIS Cut Line= 2
459206.6051048793188905.35087002 459496.043504883188734.50867002
#Sta/Elev= 30
 -203.47   12.49       0    7.85   25.07    7.05   42.91    5.79  100.41    5.56
  145.54    6.15   199.7    5.24  208.46    6.89  421.34    6.61  438.02    6.97
  446.08    8.07  452.93    5.22  453.93    5.67  472.65    3.79   526.4    3.67
   559.4    3.04  671.59    2.92  688.24    5.68  690.71       3  834.22    3.28
   849.8    3.05  869.25    1.06  890.73    2.39  925.72     3.3  945.46    2.11
 1001.21    3.36 1012.38    2.62 1022.29    6.41 1043.84    8.97 1109.23   11.16
#Mann= 3 , 0 , 0
 -203.47     .22       0  446.08      .2       0 1022.29     .22       0
Bank Sta=446.08,1022.29
XS Rating Curve= 0 ,0
Exp/Cntr=0.3,0.1

Type RM Length L Ch R = 1 ,252.74  ,5512.566,5512.566,5512.566
BEGIN DESCRIPTION:
XS4
END DESCRIPTION:
Node Name=XS4
XS GIS Cut Line= 2
 459796.085804883189458.56807002459959.3749048793189243.81887002
#Sta/Elev= 30
       0     9.9   42.39     7.6   88.08     6.4  181.08       6  199.29     4.2
  217.94       1  227.49      .9  237.53     1.6  302.16     3.4  320.12     3.1
  336.83     4.2  386.81       4  403.81     4.6  420.13     3.7  459.91     4.7
  574.87     5.1  589.66     3.1  608.16     1.9   623.7     1.8  672.08    -1.2
  681.48     2.1  710.32     1.8  744.17     2.6  815.27     2.6  831.64     3.8
  841.78     6.5  848.97     7.3  887.35     6.6  929.63     8.1 1017.41   17.39
#Mann= 5 , 0 , 0
       0     .22       0  199.29     .22       0  336.83     .22       0
  574.87      .2       0  848.97     .22       0
Bank Sta=574.87,848.97
XS Rating Curve= 0 ,0
Exp/Cntr=0.3,0.1

Type RM Length L Ch R = 1 ,197.61  ,5438.025,5438.025,5438.025
BEGIN DESCRIPTION:
XS3
END DESCRIPTION:
Node Name=XS3
XS GIS Cut Line= 2
460829.9461048793190407.87167002 461055.296404883190115.14967002
#Sta/Elev= 30
 -287.57      11   24.29    5.35   62.45    4.19  147.14    4.23  162.34    1.31
  181.07    1.23  251.16    1.75  260.17    3.79  306.92    3.47  316.45    4.95
  333.84    4.45  434.75    5.14  457.35    5.89  537.66    4.91  680.61    4.29
  696.41    5.08  700.12    3.78  713.88    2.51  749.25    1.55  763.67    2.37
  786.91    1.23  799.86     .04  820.09   -5.48  848.03     .97  882.09    5.36
   888.3    4.64   920.2    4.53 1093.85    7.23 1173.86    9.44 1219.12    9.96
#Mann= 5 , 0 , 0
 -287.57     .22       0  147.14     .22       0  260.17     .22       0
  696.41      .2       0  882.09     .22       0
#XS Ineff= 1 ,-1
   48.35  316.45    4.95
Permanent Ineff=
       T
Bank Sta=696.41,882.09
XS Rating Curve= 0 ,0
Exp/Cntr=0.3,0.1

Type RM Length L Ch R = 1 ,143.23  ,6633.826,6633.826,6633.826
BEGIN DESCRIPTION:
XS2
END DESCRIPTION:
Node Name=XS2
XS GIS Cut Line= 2
461765.1722048793191043.89447002461806.0515048793191038.38137002
#Sta/Elev= 30
 -855.27   14.47 -760.24   12.16 -570.18    7.01 -475.15    5.29 -380.12    4.53
  -95.03    3.75       0    3.72     .19    4.13       7    4.48   12.81    3.86
   21.53    2.47    31.3    1.59    50.2     .35   60.36   -1.88   69.85   -3.71
   80.05   -5.43   92.54   -5.96  101.09   -3.44  105.43   -1.23  110.62    3.06
   113.9    4.68   126.9    5.03  136.82    4.15  324.44       5  605.87    5.07
  793.49    5.46   887.3    6.04 1168.73    8.35 1262.54    9.78 1356.34   11.43
#Mann= 3 , 0 , 0
 -855.27     .22       0       7      .2       0   113.9     .22       0
#XS Ineff= 1 ,-1
 -380.12       7    4.48
Permanent Ineff=
       T
Bank Sta=7,113.9
XS Rating Curve= 0 ,0
Exp/Cntr=0.3,0.1

Type RM Length L Ch R = 1 ,76.89   ,2563,2563,2563
BEGIN DESCRIPTION:
XS1
END DESCRIPTION:
Node Name=XS1
XS GIS Cut Line= 2
 462803.448104883191969.26997002 462859.554904883191908.91657002
#Sta/Elev= 30
-4928.99   10.08 -4876.5    7.96-4699.35    3.01-4207.28    2.07 -3013.2    1.51
-1582.93       2 -684.97     4.6 -195.71    1.85       0    2.01     .13     2.8
   24.53    2.41   33.99    3.61   43.96    1.95   71.39     .67   80.11   -1.39
  104.67   -4.69  117.04    -3.2  145.01    -5.8  158.26   -4.21  173.58     .72
  191.04    1.85  201.37    3.56  212.86    2.42  236.92     2.1  270.18    2.86
  272.17    2.35  368.96    1.82 1240.11    1.95 1336.91    3.85  1433.7    7.93
#Mann= 3 , 0 , 0
-4928.99     .22       0   33.99      .2       0  201.37     .22       0
#XS Ineff= 3 ,-1
-4837.13 -684.97       7 -489.26   33.99       4  201.37 1336.91       4
Permanent Ineff=
       F       F       F
Bank Sta=33.99,201.37
XS Rating Curve= 0 ,0
Exp/Cntr=0.3,0.1

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
Type RM Length L Ch R = 1 ,0       ,7.0538,7.0538,7.0538
BEGIN DESCRIPTION:
LoWek
END DESCRIPTION:
Node Name=LoWek
XS GIS Cut Line= 2
  463445.2442725 3193619.5738227  463552.4459684 3193623.8064514
#Sta/Elev= 30
   -6800   11.97-6275.23      11-5658.62    8.87-5278.16       6-5081.38       4
-5042.02    3.04-4851.79    2.06-3001.98       2-2798.63    1.08 -522.45     .99
 -227.26       0    -130     .31    -110    -1.6     -75    -2.9     -70    -3.9
     -55   -3.55     -30    -4.4     -20    -6.1       0    -5.1       5   -1.22
      20     .18  1694.7    1.29  3420.4       4 3518.69    8.09 3715.27   10.97
 3862.71   13.96 4059.28   14.96  4403.3   15.07 4452.44   15.95  5287.9      17
#Mann= 3 , 0 , 0
   -6800     .22       0    -130      .2       0      20     .22       0
#XS Ineff= 2 ,-1
 -5284.8  -561.8       6  743.56 3518.69       6
Permanent Ineff=
       F       F
Bank Sta=-130,20
XS Rating Curve= 0 ,0
Exp/Cntr=0.3,0.1
Stream Node=LtWekiva        ,LtWekiva        , 0 , 0 ,Upstream end
Stream Node=LtWekiva        ,LtWekiva        , 0 , 1 ,Downstream end
Stream Node=ROK             ,ROK             , 0 , 0 ,Upstream end
Stream Node=ROK             ,ROK             , 0 , 1 ,Downstream end
Stream Node=wekiva          ,wek_run         , 0 , 0 ,Upstream end
Stream Node=wekiva          ,wek_run         , 0 , 1 ,Downstream end
Stream Node=wekiva          ,wekiva_riv_up   , 0 , 0 ,Upstream end
Stream Node=wekiva          ,wekiva_riv_up   , 0 , 1 ,Downstream end
Stream Node=wekiva          ,wekiva_riv_down , 0 , 0 ,Upstream end
Stream Node=wekiva          ,wekiva_riv_down , 0 , 1 ,Downstream end
LCMann Table=0

Chan Stop Cuts=-1
Use User Specified Reach Order=0
Roughness Change=ROK             ,ROK             ,160.48  ,18.07   , 5
      50       1      60     .85      75      .7     120      .6     420      .5
Roughness Change=wekiva          ,wekiva_riv_down ,544.57  ,0       , 5
     140       1     200      .8     400     .65     700    .575    2000      .5
Roughness Change=ROK             ,ROK             ,396.13  ,350.27  , 2
      46       1     120      .5
Roughness Change=LtWekiva        ,LtWekiva        ,107.56* ,30.50   , 5
      30       1      50    .773      70    .636     140    .545    1020    .455
Roughness Change=LtWekiva        ,LtWekiva        ,143.98  ,143.98  , 5
      30       1      48    .773      70    .636     120    .545     640    .455
Roughness Change=wekiva          ,wekiva_riv_up   ,678.62  ,579.64  , 5
      90       1     120      .8     200     .75     300     .65    1000      .5
Roughness Change=wekiva          ,wekiva_riv_up   ,747.29  ,711.81  , 5
      90       1     120      .8     200     .75     300     .65    1000      .5
Roughness Change=wekiva          ,wek_run         ,785.19  ,779.51  , 5
      50       1      60      .8      80     .75     100     .65     500      .5
Composite Channel Slope=5

--- wekiva_ras.g06 (geometry) ---

Geom Title=wekiva_ras_2018_ft_10
Program Version=5.03

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
Junct Name=Junc_Rok
Junct Desc=, 0 , 0 ,-1 ,0
Up River,Reach=ROK             ,ROK
Up River,Reach=wekiva          ,wek_run
Dn River,Reach=wekiva          ,wekiva_riv_up
Junc L&A=0,0
Junc L&A=0,0

River Reach=LtWekiva        ,LtWekiva

Type RM Length L Ch R = 1 ,312.14  ,6167.191,6167.191,6167.191
BEGIN DESCRIPTION:
TheSprings
END DESCRIPTION:
Node Name=TheSprings
XS GIS Cut Line= 2
461204.5570048793173492.65727002461225.0887048793173489.69387002
#Sta/Elev= 21
       0   28.92       5   28.97       7   28.76      10   28.05      15   26.22
      16   22.88      17   21.96      20   21.89      25   22.15      30   21.69
      33   22.89      34   24.57      35    24.8      40   25.28      41   25.36
      43   25.75      45   26.24      49   27.98      50   28.35      55   29.69
      59   30.83
#Mann= 3 , 0 , 0
       0     .15       0      16    .043       0      33     .15       0
Bank Sta=16,33
XS Rating Curve= 0 ,0
Exp/Cntr=0.3,0.1

Type RM Length L Ch R = 1 ,250.47  ,195.8661,195.8661,195.8661
BEGIN DESCRIPTION:
MFL_SLB_south
END DESCRIPTION:
Node Name=MFL_SLB_south
XS GIS Cut Line= 2
 461695.722804883174963.91247002461744.7818048793175039.17377002
#Sta/Elev= 30
       0  22.582      10  21.142      40  18.522      48  19.052      53  18.552
      80  18.022      90  18.312     100  17.452     111  17.692     115  18.842
     160  18.082     200  18.452     223  19.242     224  17.512   224.5  16.072
     235  15.682     240  14.672     245  15.522     250  17.532     253  19.542
     255  19.682     270  18.932     360  18.222     365  18.012   365.6  17.402
     375  17.252     390  18.762     420  18.982     430  22.202     450  24.672
#Mann= 3 , 0 , 0
       0     .15       0     223    .055       0     255     .15       0
#XS Ineff= 2 ,-1
      30     220   19.24     255     425   19.68
Permanent Ineff=
       F       F
Bank Sta=223,255
XS Rating Curve= 0 ,0
Exp/Cntr=0.3,0.1

Type RM Length L Ch R = 1 ,248.51  ,282.3819,282.3819,282.3819
BEGIN DESCRIPTION:
MFL_SLB_bridge
END DESCRIPTION:
Node Name=MFL_SLB_bridge
XS GIS Cut Line= 2
461657.0487048793175034.72957002461736.0472048793175081.44547002
#Sta/Elev= 30
       0  22.632       8  21.882     8.1  21.592      38  17.342      45  16.782
      58  17.422      65  19.222      70  18.452      75  18.882      76  17.272
      85  16.462      90  15.222      95  14.762     105  16.382     110  16.492
     118  18.392     130  19.362     150  19.582     165  19.112     185  19.252
     219  18.182     235  18.602     260  18.632     270  17.672     280  17.232
     284  17.562     285  18.452     295  18.932     305  20.722     308  20.902
#Mann= 3 , 0 , 0
       0     .15       0      65    .055       0     130     .15       0
#XS Ineff= 2 ,-1
      20      65   19.22     130     300   19.36
Permanent Ineff=
       F       F
Bank Sta=65,130
XS Rating Curve= 0 ,0
Exp/Cntr=0.3,0.1

Type RM Length L Ch R = 1 ,245.69  ,6319.948,6319.948,6319.948
BEGIN DESCRIPTION:
MFL_SLB_north
END DESCRIPTION:
Node Name=MFL_SLB_north
XS GIS Cut Line= 3
461616.7210048793175109.23877002 461714.682104883175129.98127002
462481.3654001193175292.32048682
#Sta/Elev= 30
       0  21.512      70  18.612     150  18.092     160  17.582     170  17.922
     190  17.162     200  18.032     210  17.582     215  18.282     242  19.122
     244  16.932     250  15.672     260  15.572     265  15.622     272  17.092
     275  18.622     280  18.692     305  18.252     310  17.282     330  17.662
     370  17.062     400  18.652     430  17.622     450  18.792     460  17.982
     500  18.872954.9455 19.16271148.509      23  1196.9      231293.682 24.8808
#Mann= 3 , 0 , 0
       0     .15       0     242    .055       0     280     .15       0
#XS Ineff= 2 ,-1
      60     242   19.12     280     470   18.69
Permanent Ineff=
       F       F
Bank Sta=242,280
XS Rating Curve= 0 ,0
Exp/Cntr=0.3,0.1

Type RM Length L Ch R = 1 ,182.49  ,3850.361,3850.361,3850.361
BEGIN DESCRIPTION:
MFL_Sabol
MFL_Sabol
END DESCRIPTION:
Node Name=MFL_Sabol
XS GIS Cut Line= 2
 460724.291904883176565.62067002 461198.426104883176557.15397002
#Sta/Elev= 30
-860.094      16-762.169      15-370.471 14.9302-321.509      14       0  13.668
      60  14.348      64  13.378      66  11.838      90  10.958     140  13.188
     150  13.038     160  11.458     170  12.328     180  11.278     190  12.078
     198   9.498     205   9.138     210  11.838     220  11.488     230  13.768
     244  13.618     245  12.688     250  10.618     255  11.818     260  11.988
     266  14.778363.9624 15.0659412.9247 15.9882559.8115 17.1129755.6606 20.9429
#Mann= 3 , 0 , 0
-860.094     .15       0     190    .055       0     210     .15       0
#XS Ineff= 1 ,-1
      64     120   12.08
Permanent Ineff=
       F
Bank Sta=190,210
XS Rating Curve= 0 ,0
Exp/Cntr=0.3,0.1

Type RM Length L Ch R = 1 ,143.98  ,3642.73,3642.73,3642.73
BEGIN DESCRIPTION:
LW2
END DESCRIPTION:
Node Name=LW2
XS GIS Cut Line= 2
 460933.299004883177665.03007002461212.6995048793177544.37987002
#Sta/Elev= 30
   -6000      15       0  11.086     300  11.586     500  12.286   501.5  12.006
     505  11.986     525   9.386     530   9.086     535   8.386     540   7.986
     555   7.986     560   8.786     565   8.486     570   9.086     575   9.086
     580   8.386     595   9.686     600   9.486     607  12.486     707  11.886
     807  11.486    1107  11.7862032.791      142131.163      152180.349  15.072
2229.535 15.99112327.908      162377.094 16.7483 2426.28      172524.652      18
#Mann= 3 , 0 , 0
   -6000       0       0     500       0       0     607       0       0
#XS Ineff= 2 ,-1
   -2000     500   12.29     607    1400   12.49
Permanent Ineff=
       F       F
Bank Sta=500,607
XS Rating Curve= 0 ,0
Vertical n Elevations= 5
      30      48      70     120     640
Vertical n for Station=-6000
     .22     .22     .22     .22     .22
Vertical n for Station=500
      .2     .17     .14     .12      .1
Vertical n for Station=607
     .22     .22     .22     .22     .22
Vertical n Flow=-1
Exp/Cntr=0.3,0.1

Type RM Length L Ch R = 1 ,71.13   ,4063.156,4063.156,4063.156
BEGIN DESCRIPTION:
LW1
END DESCRIPTION:
Node Name=LW1
XS GIS Cut Line= 2
460177.6475048793179246.18327002 460425.298004883179284.28337002
#Sta/Elev= 30
-2170.99      14-2111.97      14-2085.74 13.0294-1967.72 12.9532-1895.59      12
     100  11.522     200  11.022     400  11.022     500  11.942     507  10.042
     517   9.042     522   9.142     532   8.142     547   7.742     552   8.342
     572   8.642     577   9.342     592   9.642     597  10.542     601  12.442
     700  10.842    1100  11.3421655.207      141704.387 14.27811753.567 14.9583
1999.466 15.02082097.825      162294.545 16.02972343.725 16.70992442.084      17
#Mann= 3 , 0 , 0
-2170.99       0       0     500       0       0     601       0       0
#XS Ineff= 2 ,-1
-1226.79     500   11.94     601    1350   12.44
Permanent Ineff=
       F       F
Bank Sta=500,601
XS Rating Curve= 0 ,0
Vertical n Elevations= 5
      30      50      70     140    1020
Vertical n for Station=-2170.99
     .22     .22     .22     .22     .22
Vertical n for Station=500
      .2     .17     .14     .12      .1
Vertical n for Station=601
     .22     .22     .22     .22     .22
Vertical n Flow=-1
Exp/Cntr=0.3,0.1

Type RM Length L Ch R = 1 ,30.50   ,3049.836,3049.836,3049.836
BEGIN DESCRIPTION:
WK18
END DESCRIPTION:
Node Name=WK18
XS GIS Cut Line= 2
 459515.919704883180360.70577002 459987.937304883180315.19737002
#Sta/Elev= 30
 -206.62      13-180.390 12.0255-108.269 11.9891-88.6005  11.765-3.36730 11.9961
       0  11.422     100  11.522     200  11.022     300  11.222     400  11.022
     500  11.283     515  11.023     520   9.653     525   6.753     530   6.053
     540   5.653     545   6.853     550   6.653     555   6.753     565   8.353
     571  10.293     573  11.663     575  11.323     601  12.442     700  10.842
    1100  11.3421294.801      111825.869 10.7326 3125.62 14.38723174.641      15
#Mann= 3 , 0 , 0
 -206.62       0       0     500       0       0     601       0       0
#XS Ineff= 2 ,-1
     100     500   11.28     601    2450   12.44
Permanent Ineff=
       F       F
Bank Sta=500,601
XS Rating Curve= 0 ,0
Vertical n Elevations= 5
      30      50      70     140    1020
Vertical n for Station=-206.62
     .22     .22     .22     .22     .22
Vertical n for Station=500
      .2     .17     .14     .12      .1
Vertical n for Station=601
     .22     .22     .22     .22     .22
Vertical n Flow=-1
Exp/Cntr=0.3,0.1

River Reach=ROK             ,ROK

Type RM Length L Ch R = 1 ,480.77  ,149.0814,149.0814,149.0814
BEGIN DESCRIPTION:
RokSpr02
END DESCRIPTION:
Node Name=RokSpr02
XS GIS Cut Line= 2
451026.6781048793181095.07657002451022.5373048793181071.37427002
#Sta/Elev= 30
       0  28.228       2  29.928       4  27.558       5  25.928       6  22.988
       8  23.928      10  23.648      12  24.008      14  22.848      18  22.948
      20  24.208      22  24.128      24  24.618      30  24.628      32  24.608
      34  24.418      36  23.388      38  23.578      42  23.608      46  22.908
      48  22.718      50  23.178      52  23.348      54  23.818      58  23.558
      62  23.928      65  24.708      66  25.918      68  27.798   76.19  29.928
#Mann= 3 , 0 , 0
       0     .15       0       5     .04       0      66     .15       0
Bank Sta=5,66
XS Rating Curve= 0 ,0
Exp/Cntr=0.3,0.1

Type RM Length L Ch R = 1 ,479.28  ,145.1115,145.1115,145.1115
BEGIN DESCRIPTION:
RokSpr03
END DESCRIPTION:
Node Name=RokSpr03
XS GIS Cut Line= 2
451082.3677048793181066.28987002451051.4643048793181054.43647002
#Sta/Elev= 24
       0  27.218       5  26.668       8  25.888       9  25.418      12  24.898
      14  24.138      15  23.898      16  23.218      18  22.678      20  22.428
      22  22.398      23  22.548      24  22.598      26  22.968      27  23.318
      28  23.938      29  23.828      31  23.998      32  24.158      34  24.918
      35  25.058      36  25.508      38  25.878      39  26.288
#Mann= 3 , 0 , 0
       0     .15       0      12     .04       0      34     .15       0
Bank Sta=12,34
XS Rating Curve= 0 ,0
Exp/Cntr=0.3,0.1

Type RM Length L Ch R = 1 ,477.83  ,396.8176,396.8176,396.8176
BEGIN DESCRIPTION:
RokSpr04
END DESCRIPTION:
Node Name=RokSpr04
XS GIS Cut Line= 2
 451097.184404883181024.59137002 451068.609404883181013.79637002
#Sta/Elev= 28
       0  26.448       7  26.338      11  25.678      12  25.078      14  24.628
      15  24.528      16  24.648      17  24.608      20  24.088      22  23.498
      23  22.698      25  22.598      26  22.878      27  22.958      28  23.168
      29  23.538      31  23.888      33  23.638      34  23.858      35  23.818
      36  23.878      37  24.038      38  23.918      40  24.398      41  24.758
      43  25.088      45  25.368      47  26.078
#Mann= 3 , 0 , 0
       0     .15       0      12     .04       0      43     .15       0
Bank Sta=12,43
XS Rating Curve= 0 ,0
Exp/Cntr=0.3,0.1

Type RM Length L Ch R = 1 ,473.86  ,436.3189,436.3189,436.3189
BEGIN DESCRIPTION:
RokSpr05
END DESCRIPTION:
Node Name=RokSpr05
XS GIS Cut Line= 2
451175.4950048793180987.69237002451172.3109048793180957.39027002
#Sta/Elev= 30
       0  26.818       4  25.028      10  24.308      15  24.838      19  24.638
      25  24.228      26  23.768      27  23.828      28  23.468      30  23.588
      31  24.048      32  23.848      34  24.048      38  23.868      41  23.168
      44  23.098      46  22.698      50  22.658      56  23.638      58  23.308
      61  23.408      65  23.188      68  23.828      70  24.528      74  24.808
      75  25.118      79  24.688      80  25.008      90  25.498     100  26.798
#Mann= 3 , 0 , 0
       0     .15       0       4     .04       0      75     .15       0
Bank Sta=4,75
XS Rating Curve= 0 ,0
Exp/Cntr=0.3,0.1

Type RM Length L Ch R = 1 ,469.5   ,86.1877,86.1877,86.1877
BEGIN DESCRIPTION:
RokSpr08
END DESCRIPTION:
Node Name=RokSpr08
XS GIS Cut Line= 2
 451256.572004883181058.88917002451286.3376048793181034.67977002
#Sta/Elev= 21
       0  27.608       1  25.318     1.1  22.088       2  21.988       4  21.938
       8  22.068      16  21.938      24  21.968      38  21.818      48  21.918
      52  22.108      56  22.698      58  22.848      60  23.518      62  23.268
      64  23.618      68  23.898      74  24.568      76  25.328      80  26.768
   80.46  26.768
#Mann= 3 , 0 , 0
       0     .15       0       1     .04       0      76     .15       0
Bank Sta=1,76
XS Rating Curve= 0 ,0
Exp/Cntr=0.3,0.1

Type RM Length L Ch R = 1 ,468.64  ,242.6181,242.6181,242.6181
BEGIN DESCRIPTION:
RokSpr09
END DESCRIPTION:
Node Name=RokSpr09
XS GIS Cut Line= 2
 451276.415704883181079.12987002 451298.510204883181052.33677002
#Sta/Elev= 17
       0  26.048     1.5  25.308     1.5  21.708       4  21.858       6  21.678
      16  21.608      32  21.858      40  22.168      44  22.488      50  23.358
      58  23.808      62  24.158      66  24.848      67  25.308      70  26.608
      75  27.338   75.56  27.338
#Mann= 3 , 0 , 0
       0     .15       0     1.5     .04       0      67     .15       0
Bank Sta=1.5,67
XS Rating Curve= 0 ,0
Exp/Cntr=0.3,0.1

Type RM Length L Ch R = 1 ,466.21  ,193.2415,193.2415,193.2415
BEGIN DESCRIPTION:
RokSpr11
END DESCRIPTION:
Node Name=RokSpr11
XS GIS Cut Line= 2
451331.5027048793181121.98737002 451349.007504883181107.29797002
#Sta/Elev= 30
       0  26.768       5  26.988      10  26.778      15  26.948      20  26.838
      27  27.078      29  25.238      30  24.898      32  24.618      36  23.768
      40  22.588      41  22.408      42  22.578      45  22.128      48  22.208
      50  22.128      53  22.228      56  22.908      58  22.768      59  22.558
      60  22.578      62  22.398      64  22.558      66  22.888      67  22.858
      68  23.018      70  23.768      71  25.198      72  26.178      75  26.568
#Mann= 3 , 0 , 0
       0     .15       0      36     .04       0      70     .15       0
Bank Sta=36,70
XS Rating Curve= 0 ,0
Exp/Cntr=0.3,0.1

Type RM Length L Ch R = 1 ,464.28  ,196.4567,196.4567,196.4567
BEGIN DESCRIPTION:
RokSpr12
END DESCRIPTION:
Node Name=RokSpr12
XS GIS Cut Line= 2
 451376.887304883181161.36027002 451390.891104883181147.35337002
#Sta/Elev= 30
       0  25.828       7  25.838       9  25.168     9.1  24.778      10  24.438
      13  23.648      18  22.788      20  22.768      21  22.518      23  22.488
      25  21.638      26  21.518      34  21.578      39  22.398      40  22.348
      42  22.628      43  22.888      46  23.008      49  23.538      50  23.558
      51  24.028      53  23.818      54  23.868      56  24.458      57  24.488
      59  24.878      60  24.878      61  25.188      62  26.218      65  26.768
#Mann= 3 , 0 , 0
       0     .15       0      20     .04       0      43     .15       0
Bank Sta=20,43
XS Rating Curve= 0 ,0
Exp/Cntr=0.3,0.1

Type RM Length L Ch R = 1 ,462.31  ,239.5341,239.5341,239.5341
BEGIN DESCRIPTION:
RokSpr13
END DESCRIPTION:
Node Name=RokSpr13
XS GIS Cut Line= 2
451422.9117048793181205.33417002 451436.623104883181181.58607002
#Sta/Elev= 30
       0  25.828      25  25.988      29  25.148      30  24.508      32  24.608
      38  24.428      42  24.098      44  23.698      45  23.818      46  23.688
      47  23.298      48  23.028      51  22.748      52  22.228      53  22.148
      55  21.538      57  21.508      60  21.648      61  21.828      62  22.268
      65  22.498      68  23.388      76  23.598      78  23.248      79  23.368
      81  24.498      83  24.828      85  25.568      88  26.388      90  26.608
#Mann= 3 , 0 , 0
       0     .15       0      47     .04       0      68     .15       0
Bank Sta=47,68
XS Rating Curve= 0 ,0
Exp/Cntr=0.3,0.1

Type RM Length L Ch R = 1 ,459.92  ,1057.185,1057.185,1057.185
BEGIN DESCRIPTION:
RokSpr14
END DESCRIPTION:
Node Name=RokSpr14
XS GIS Cut Line= 2
451484.9297048793181229.40207002 451504.259604883181220.38617002
#Sta/Elev= 30
       0  26.008       3  25.808       5  25.088       7  24.808      10  24.608
      16  24.438      17  24.278      19  23.768      20  23.428      21  22.868
      22  22.858      25  22.508      32  22.348      34  22.018      35  21.998
      38  22.238      41  22.688      44  22.928      45  23.128      48  22.588
      52  22.378      54  22.368      56  22.568      57  22.758      58  23.818
      59  24.598      60  24.438      61  24.698      67  26.678      70  26.078
#Mann= 3 , 0 , 0
       0     .15       0      19     .04       0      58     .15       0
Bank Sta=19,58
XS Rating Curve= 0 ,0
Exp/Cntr=0.3,0.1

Type RM Length L Ch R = 1 ,449.35  ,5321.588,5321.588,5321.588
BEGIN DESCRIPTION:
ROK7
END DESCRIPTION:
Node Name=ROK7
XS GIS Cut Line= 2
 451531.470204883181508.48117002 451753.720604883181451.33097002
#Sta/Elev= 30
    1969    28.9    1997    28.9    2000    28.4    2006    23.8    2015    23.1
    2016    20.2    2020    20.1    2025    20.5    2035    22.9    2050    22.9
    2055    23.6    2060    23.1    2085    23.9    2115    22.9    2125    23.5
    2135    23.5    2138   23.75    2143    25.1    2171    23.8    2173    23.3
    2177    23.2    2183    23.8    2185    24.9    2200    24.4    2300    23.9
    2400    24.9    2500    24.8    2600    25.3    2650      24    3000    28.9
#Mann= 3 , 0 , 0
    1969     .18       0    2006     .04       0    2085     .18       0
Bank Sta=2006,2085
XS Rating Curve= 0 ,0
Exp/Cntr=0.3,0.1

Type RM Length L Ch R = 1 ,396.13  ,4586.122,4586.122,4586.122
BEGIN DESCRIPTION:
ROK6
END DESCRIPTION:
Node Name=ROK6
XS GIS Cut Line= 2
450737.7186048793182638.78337002451099.6693048793182740.38357002
#Sta/Elev= 30
    1950   23.91    2000   23.11    2002   21.71    2005   21.31    2015   20.61
    2020   19.81    2025   19.71    2030   20.21    2035   19.51    2040   19.51
    2045   18.91    2050   18.61    2060   18.81    2065   20.01    2070   19.81
    2075   19.31    2080   19.31    2085   19.61    2090   19.21    2100   19.11
    2105   19.91    2110   20.51    2115   20.81  2127.5   22.51    2150   21.81
    2300   21.81    2400   22.31    2500   21.91    2600   23.41    2630   23.61
#Mann= 3 , 0 , 0
    1950     .18       0    2000      .2       0  2127.5     .18       0
Bank Sta=2000,2127.5
XS Rating Curve= 0 ,0
Vertical n Elevations= 5
      46      49      51      54     120
Vertical n for Station=1950
     .22     .22     .22     .22     .22
Vertical n for Station=2000
      .2     .17     .14     .12      .1
Vertical n for Station=2127.5
     .22     .22     .22     .22     .22
Vertical n Flow=-1
Exp/Cntr=0.3,0.1

Type RM Length L Ch R = 1 ,350.27  ,13446.29,13446.29,13446.29
BEGIN DESCRIPTION:
ROK5
END DESCRIPTION:
Node Name=ROK5
XS GIS Cut Line= 2
 451861.670804883183629.38537002 451766.420704883183273.78467002
#Sta/Elev= 30
     900   23.92    1500   20.62    1700   21.42    1800   20.92    1900   21.02
    2000   22.02  2003.5   20.63    2005   19.82    2010   19.42    2025   19.02
    2035   19.02    2040   19.22    2055   19.42    2065   19.32    2075   19.02
    2085   19.42    2095   19.12    2105   19.42    2125   19.12    2140   19.32
    2150   19.02    2155   19.12    2160   19.92    2165   21.12    2220   21.32
    2300   21.02    2400   21.22    2600   20.82    2665   21.02    4500   23.92
#Mann= 3 , 0 , 0
     900     .18       0    2000      .2       0    2220     .18       0
Bank Sta=2000,2220
XS Rating Curve= 0 ,0
Vertical n Elevations= 5
      46      49      51      54     120
Vertical n for Station=900
     .22     .22     .22     .22     .22
Vertical n for Station=2000
      .2     .17     .14     .12      .1
Vertical n for Station=2220
     .22     .22     .22     .22     .22
Vertical n Flow=-1
Exp/Cntr=0.3,0.1

Type RM Length L Ch R = 1 ,215.81  ,5532.677,5532.677,5532.677
BEGIN DESCRIPTION:
ROK4
END DESCRIPTION:
Node Name=ROK4
XS GIS Cut Line= 2
 453798.424704883181095.73027002453442.8240048793181038.58017002
#Sta/Elev= 30
  1257.5   23.94    1300   23.44    1600   20.74    1700   20.04    1800   20.04
    1900   20.54    2000   20.54    2002   19.94    2007   19.32    2010   19.14
    2015   17.34    2020   16.14    2025   15.24    2030   15.44    2035   16.04
    2040   15.34    2050   14.74    2055   14.84    2060   17.44    2064   18.64
    2070   21.34    2100   20.74    2200   20.34    2300   20.44    2400   19.84
    2500   19.84    2600   19.64    2900   21.04    3000   20.94    4000   23.94
#Mann= 3 , 0 , 0
  1257.5     .18       0    2000      .2       0    2070     .18       0
Bank Sta=2000,2070
XS Rating Curve= 0 ,0
Vertical n Elevations= 5
      48      51      55      60     250
Vertical n for Station=1257.5
     .22     .22     .22     .22     .22
Vertical n for Station=2000
      .2     .17     .14     .12      .1
Vertical n for Station=2070
     .22     .22     .22     .22     .22
Vertical n Flow=-1
Exp/Cntr=0.3,0.1

Type RM Length L Ch R = 1 ,160.48  ,3360.203,3360.203,3360.203
BEGIN DESCRIPTION:
ROK3
END DESCRIPTION:
Node Name=ROK3
XS GIS Cut Line= 2
 453683.837304883179720.61477002 453618.766804883179618.24147002
#Sta/Elev= 30
       0  23.645      20  22.545      70  21.965     100  21.175     120  19.985
     130  19.045     150  18.665     160  17.585     170  17.735     177  18.665
     190  18.755     192  18.685     193  18.175     200  17.085     215  17.485
     225  16.685     230  16.785     235  16.185     245  15.985     255  17.585
   255.5  18.685     256  18.945     270  19.005     300  18.375     320  18.555
     340  19.125     360  20.185     400  21.335     410  21.295     419  21.855
#Mann= 3 , 0 , 0
       0     .18       0     190      .2       0     256     .18       0
Bank Sta=190,256
XS Rating Curve= 0 ,0
Vertical n Elevations= 5
      50      60      75     120     420
Vertical n for Station=0
     .22     .22     .22     .22     .22
Vertical n for Station=190
      .2     .17     .14     .12      .1
Vertical n for Station=256
     .22     .22     .22     .22     .22
Vertical n Flow=-1
Exp/Cntr=0.3,0.1

Type RM Length L Ch R = 1 ,126.88  ,7053.478,7053.478,7053.478
BEGIN DESCRIPTION:
ROK2
END DESCRIPTION:
Node Name=ROK2
XS GIS Cut Line= 2
454544.9803048793179351.14227002 454484.226104883179114.52637002
#Sta/Elev= 30
    -100  22.173     -10  20.943       0  21.223      10  20.383      19  20.833
    23.5  18.893      30  18.163      40  19.693      50  19.783      90  19.153
      96  18.063     103  19.173     150  19.153     210  18.493     240  17.233
     280  17.243     310  18.013     363  17.453     371  14.563     375  14.403
     385  14.553     410  16.613     430  15.163     450  17.023     520  17.263
     540  18.533     560  18.923     570  17.643     580  19.883     587  20.703
#Mann= 3 , 0 , 0
    -100     .18       0     363      .2       0     450     .18       0
Bank Sta=363,450
XS Rating Curve= 0 ,0
Vertical n Elevations= 5
      50      60      75     120     420
Vertical n for Station=-100
     .22     .22     .22     .22     .22
Vertical n for Station=363
      .2     .17     .14     .12      .1
Vertical n for Station=450
     .22     .22     .22     .22     .22
Vertical n Flow=-1
Exp/Cntr=0.3,0.1

Type RM Length L Ch R = 1 ,56.34   ,3817.881,3817.881,3817.881
BEGIN DESCRIPTION:
ROK1
END DESCRIPTION:
Node Name=ROK1
XS GIS Cut Line= 2
455779.6287048793178130.27437002455392.2779048793178035.02417002
#Sta/Elev= 30
     500   18.97    2500   15.97    2600   15.17    2800   14.67    2819   14.47
    2840   13.47    2857   13.47    2861   14.57    3000   14.97    3003   13.77
    3045   13.17    3050   12.67    3065   13.37    3080   12.77    3100   13.77
    3103   13.47    3105   11.27    3110   10.47    3124   11.07    3132   13.37
    3135   13.47    3160   12.57    3182   13.37    3185   15.57    3234   14.27
    3245   13.57    3271   13.77    3273   14.17    3685   13.67    6400   18.97
#Mann= 3 , 0 , 0
     500     .18       0    3100      .2       0    3135     .18       0
Bank Sta=3100,3135
XS Rating Curve= 0 ,0
Vertical n Elevations= 5
      50      60      75     120     420
Vertical n for Station=500
     .22     .22     .22     .22     .22
Vertical n for Station=3100
      .2     .17     .14     .12      .1
Vertical n for Station=3135
     .22     .22     .22     .22     .22
Vertical n Flow=-1
Exp/Cntr=0.3,0.1

Type RM Length L Ch R = 1 ,18.17   ,1816.503,1816.503,1816.503
BEGIN DESCRIPTION:
WK16
END DESCRIPTION:
Node Name=WK16
XS GIS Cut Line= 2
 456154.279404883176999.97207002455735.1786048793176961.87207002
#Sta/Elev= 23
       0   18.98    3000   16.98    4800   15.98    7000   12.08    7025   11.98
    7050   11.78    7075   12.28    7095   11.98    7100   11.28    7105    8.58
    7110    7.68    7125   10.18    7130    8.58    7135    7.78    7140    9.88
    7150   10.38    7165   12.08    7185   11.78    7210   11.68    7235   11.18
    7260   11.28    7285   11.28   11800   18.98
#Mann= 3 , 0 , 0
       0     .18       0    7075      .2       0    7165     .18       0
Bank Sta=7075,7165
XS Rating Curve= 0 ,0
Vertical n Elevations= 5
      50      60      75     120     420
Vertical n for Station=0
     .22     .22     .22     .22     .22
Vertical n for Station=7075
      .2     .17     .14     .12      .1
Vertical n for Station=7165
     .22     .22     .22     .22     .22
Vertical n Flow=-1
Exp/Cntr=0.3,0.1

River Reach=wekiva          ,wek_run

Type RM Length L Ch R = 1 ,793.32  ,813.0906,813.0906,813.0906
BEGIN DESCRIPTION:
WekSpr6
WekSpr6
END DESCRIPTION:
Node Name=WekSpr6
XS GIS Cut Line= 2
     455071.1753     3176243.645     455098.0644     3176211.408
#Sta/Elev= 30
       6   13.22       8   13.13     8.5   11.78       9    8.47      10    8.43
      11     8.6      13    9.16      14    8.49      15    8.93      16    8.75
      17    9.19      18    9.32      22    9.45      24    9.76      25    9.76
      26      10      29   10.22      30   10.45      38    10.7      42   10.64
      43   10.79      45   10.61      53   10.62      57   10.02      65    9.29
      66    9.31      75    8.26      76    8.27    76.5   11.77      79   11.97
#Mann= 5 ,-1 , 0
       6     .22       0     8.5     .17       0      26     .22       0
      57     .17       0    76.5     .22       0
Bank Sta=8.5,76.5
XS Rating Curve= 0 ,0
Exp/Cntr=0.3,0.1

Type RM Length L Ch R = 1 ,785.19  ,567.8806,567.8806,567.8806
BEGIN DESCRIPTION:
WEK13
END DESCRIPTION:
Node Name=WEK13
XS GIS Cut Line= 2
 455163.677404883176530.07117002455328.7778048793176295.12067002
#Sta/Elev= 30
    1940   18.99    2280   15.99    4300   13.99    5000   11.99    6000   10.59
    6075   11.19    6090   12.19    6100   10.59    6105    8.59    6130    7.69
    6190    7.79    6210    7.49    6220    7.69    6230    7.39    6240    7.69
    6250    7.69    6280    7.39    6300    7.49    6320    6.99    6330    7.69
    6350    8.29    6365    8.99    6375   11.69    6445   11.09    6470   11.29
    6920   11.99    7800   13.99    9080   15.99    9980   17.99   10010   18.99
#Mann= 3 , 0 , 0
    1940     .22       0    6090      .2       0    6375     .22       0
Bank Sta=6090,6375
XS Rating Curve= 0 ,0
Exp/Cntr=0.3,0.1

Type RM Length L Ch R = 1 ,779.51  ,3231.857,3231.857,3231.857
BEGIN DESCRIPTION:
WK17
END DESCRIPTION:
Node Name=WK17
XS GIS Cut Line= 2
      455414.687     3176429.959      455415.957     3176385.507
#Sta/Elev= 28
     200   18.97    5700   14.67    5830   13.67    5960   12.67    6000   12.17
    6025   12.27    6050   12.47    6075   12.17    6095   12.57    6100   11.47
    6105   10.57    6110    9.77    6120    8.67    6130    8.37    6140    7.87
    6160    8.67    6170    8.17    6180    8.77    6190    8.87    6200    8.47
    6220   11.47    6230   13.37    6240   12.77    6270   12.07    6290   12.17
    6320   11.87    6340   11.97    7300   18.97
#Mann= 3 , 0 , 0
     200     .22       0    6095      .2       0    6230     .22       0
Bank Sta=6095,6230
XS Rating Curve= 0 ,0
Exp/Cntr=0.3,0.1

River Reach=wekiva          ,wekiva_riv_up

Type RM Length L Ch R = 1 ,747.19  ,799,799,799
BEGIN DESCRIPTION:
WEK12
END DESCRIPTION:
Node Name=WEK12
XS GIS Cut Line= 2
456440.0300048793176549.12117002 456224.129604883176390.37087002
#Sta/Elev= 30
     600   18.97    2600   16.97    4530   15.97    6600   11.27    7000   11.87
    7017    7.87    7022    8.57    7032    7.57    7067    9.17    7077    9.07
    7082    8.67    7092    9.17    7097    8.87    7102    9.57    7107    8.37
    7117    8.87    7132    8.77    7137    9.97    7142   10.27    7147   11.48
  7153.5   11.87    7203   12.07  7203.5   11.41    7208    9.87    7228    9.17
    7238    9.97    7248   10.17    7259   12.07    7759   11.37    8400   18.97
#Mann= 3 , 0 , 0
     600     .22       0    7000      .2       0    7259     .22       0
Bank Sta=7000,7259
XS Rating Curve= 0 ,0
Exp/Cntr=0.3,0.1

Type RM Length L Ch R = 1 ,739.30  ,50,50,50
BEGIN DESCRIPTION:
interpolation of WEK12 amd WK15
END DESCRIPTION:
#Sta/Elev= 30
       0      13  19.669   13.09  52.451  14.527   72.12  16.109  98.345  20.257
  118.01  20.907 119.465   13.25 134.331   12.73 164.063    9.59 181.465    6.52
 196.465    2.87 201.465    3.57 211.465    2.57 246.465    4.17 261.465    3.67
 276.465    3.87 281.465    4.57 286.465    3.37 311.465    3.77 326.465    6.48
 332.965    9.59 362.697   12.73 377.563   13.25  380.83  20.901 625.468  20.908
 723.322      19 967.956  19.2011114.737  22.3661212.591  26.5151310.444   31.48
#Mann= 3 , 0 , 0
       0     .22       0  118.01     .17       0  380.83     .22       0
#XS Ineff= 1 ,-1
       0  118.01      20
Permanent Ineff=
       F
Bank Sta=118.01,380.83
XS Rating Curve= 0 ,0
Exp/Cntr=0.3,0.1

Type RM Length L Ch R = 3 ,739     ,,,
Bridge Culvert--1,0,-1,-1, 0
Deck Dist Width WeirC Skew NumUp NumDn MinLoCord MaxHiCord MaxSubmerge Is_Ogee
10,30,2.6,0, 2, 2, , , 0.98, 0, 0,0,,
     118   380.9
      21      21
   17.75   17.75
     118   380.9
      21      21
   17.75   17.75
Pier Skew, UpSta & Num, DnSta & Num=  ,170.5, 2 ,170.5, 2 , 0 , 0 , 0 ,,
       1       1
       0      21
       1       1
       0      21
Pier Skew, UpSta & Num, DnSta & Num=  ,223, 2 ,223, 2 , 0 , 0 , 0 ,,
       1       1
       0      21
       1       1
       0      21
Pier Skew, UpSta & Num, DnSta & Num=  ,275.5, 2 ,275.5, 2 , 0 , 0 , 0 ,,
       1       1
       0      21
       1       1
       0      21
Pier Skew, UpSta & Num, DnSta & Num=  ,328, 2 ,328, 2 , 0 , 0 , 0 ,,
       1       1
       0      21
       1       1
       0      21
BR Coef=-1 , 0 , 0 ,, 0 ,,,0.8,-1,,0,
WSPro=,,,, 1 ,,,, 0 ,,,, 0 ,,,,-1 ,-1 ,-1 , 0 , 0 , 0 , 0 , 0
BC Design=,, 0 ,, 0 ,,,,,,
BC Use User HTab Curves=0
BC User HTab FreeFlow(D)= 0
